--- ELSEYRN.prj (project) ---

Proj Title=ELSEYRN
Current Plan=p01
Geom File=g01
Flow File=f01
Plan File=p01
DSS Export Rating Curves=0
DSS Export Rating Curve Sorted=0
DSS Export Volume Flow Curves=0
DXF OffsetX=0
DXF OffsetY=0
DXF ScaleX=0
DXF ScaleY=0

--- ELSEYRN.p01 (plan) ---

Plan Title=Floodplain
Program Version=4.00
Geom File=g01
Flow File=f01
K Sum by GR=0
Std Step Tol=0.01
Critical Tol=0.01
Num of Std Step Trials=20
Max Error Tol=0.3
Flow Tol Ratio=0.001
Split Flow NTrial=30
Split Flow Tol=0.02
Split Flow Ratio=0.02
Log Output Level=0
Friction Slope Method=1
Unsteady Friction Slope Method=2
Unsteady Bridges Friction Slope Method=1
Global Log Level=0
CheckData=False
Run HTab=0
Run UNet=0
Run PostProcess=0
UNET Theta=0
UNET Theta Warmup=0
UNET ZTol=0
UNET ZSATol=0
UNET MxIter=0
UNET MaxInSteps=0
UNET DtIC=0
UNET DtMin=0
UNET MaxCRTS=0
UNET WFStab=0
UNET SFStab=0
UNET WFX=0
UNET SFX=0
UNET DSS MLevel=0
UNET DZMax Abort=0
UNET Convert EG Bridges=0
UNET Use Existing IB Tables=0
UNET Froude Limit=0
UNET Froude Power=0
Write IC File=0
Echo Input=False
Echo Output=False
Write Detailed=0

--- ELSEYRN.f01 (steady flow) ---

Flow Title=NFF Regression Equation
Program Version=4.10
Number of Profiles= 1
Profile Names=P100yr
River Rch & RM=ELSEYRN,Main            ,22016.6
587.5026
River Rch & RM=ELSEYRN,Main            ,21111.4
593.9267
River Rch & RM=ELSEYRN,Main            ,19323.5
659.3418
River Rch & RM=ELSEYRN,Main            ,18432.2
850.9707
River Rch & RM=ELSEYRN,Main            ,18432.2
688.2391
River Rch & RM=ELSEYRN,Main            ,14219.1
895.9497
River Rch & RM=ELSEYRN,Main            ,13876.3
1000.236
River Rch & RM=ELSEYRN,Main            ,9012.1
 1080.57
River Rch & RM=ELSEYRN,Main            ,4434.6
1190.966
River Rch & RM=ELSEYRN,Main            ,246.6
1291.531
Boundary for River Rch & Prof#=ELSEYRN,Main            , 1
Up Type= 0
Dn Type= 3
Dn Slope=0.0316
DSS Import GetInterval= 0
DSS Import GetPeak= 0
DSS Import FillOption= 0

--- ELSEYRN.g01 (geometry) ---

Geom Title=USGS 10m DEM
Program Version=4.10

River Reach=ELSEYRN         ,Main
Reach XY= 30
       1947344.1      351841.095     1946652.328      352137.209
     1946101.705      352628.351     1945632.315      352301.807
     1945458.509      352342.376      1945200.91      352853.566
     1945336.498      353669.962     1945067.364      354256.184
     1944853.167      354473.745     1944139.315      354525.224
     1943977.263      354810.992     1943614.187      355004.708
     1942877.753      354845.842     1942878.232      355125.819
     1943151.669      355533.371     1943003.212      355862.759
     1942454.328      355402.742     1941367.359      355607.473
     1940845.663      355486.381     1940025.996      355592.673
      1939811.67      355421.909     1939414.731      355676.312
     1937113.069      355571.262     1936407.544      355984.036
     1935458.934      356227.984      1933377.44      356032.027
     1932863.671       356384.46     1931833.163      356290.365
      1930681.69      356626.505     1930248.887      356545.904

Type RM Length L Ch R = 1 ,22016.6 ,572.1,565,560.2
XS GIS Cut Line= 2
      1947313.94      351709.501     1947358.211      351969.918
#Sta/Elev= 30
       0 2300.63     9.8 2299.86    19.6 2299.26    29.4 2298.82    39.1 2298.53
    48.9 2298.32    58.7 2298.05    68.5 2297.64    78.3 2297.14      88 2296.65
    97.8  2296.2   107.6 2295.23   117.4  2293.3   127.2 2291.58   128.9  2291.5
     137 2291.09   143.9 2291.93   146.8 2292.28   156.5 2295.92   166.3 2301.21
   176.1    2306   185.9 2309.73   195.7 2312.95   205.4 2315.86   215.2 2318.37
     225 2320.44   234.8 2322.31   244.6  2324.1   254.4 2325.91   264.2  2327.9
#Mann= 3 , 0 , 0
       0      .1       0   127.2    .045       0   143.9      .1       0
Bank Sta=127.2,143.9
XS Rating Curve= 0 ,0
Exp/Cntr=0.3,0.1

Type RM Length L Ch R = 1 ,21451.6 ,349.8,340.2,330.6
XS GIS Cut Line= 2
     1946785.294      351943.876     1946892.065       352165.23
#Sta/Elev= 28
       0 2294.69     9.8    2291    19.7 2287.41    29.5 2284.14    39.3 2281.69
    49.2 2280.43      59 2279.59    68.8 2278.91    78.6  2278.3    88.5 2277.65
    98.3 2276.77   103.2 2276.29   108.1 2275.81     118 2275.34   118.2 2275.35
   127.8 2275.89   137.6 2277.22   147.5 2279.19   157.3 2283.08   167.1 2288.31
     177 2292.81   186.8 2296.44   196.6 2299.74   206.4 2302.97   216.3 2306.46
   226.1 2310.29   235.9 2314.32   245.8 2318.39
#Mann= 3 , 0 , 0
       0      .1       0   103.2    .045       0   127.8      .1       0
Bank Sta=103.2,127.8
XS Rating Curve= 0 ,0
Exp/Cntr=0.3,0.1

Type RM Length L Ch R = 1 ,21111.4 ,445.2,454.2,462.3
XS GIS Cut Line= 2
     1946467.586      352160.022     1946670.711      352329.293
#Sta/Elev= 30
       0 2312.07     9.8  2306.6    19.6  2301.1    29.4 2295.52    39.2 2290.15
      49 2284.75    58.8 2279.61    68.6 2274.76    78.3 2270.26    88.1 2267.42
    97.9 2266.18   107.7 2265.68   112.4 2265.61   117.5 2265.54   127.3    2266
   127.4 2266.01   137.1 2266.84   146.9  2267.7   156.7 2268.45   166.5 2269.17
   176.3  2269.9   186.1 2270.67   195.9 2271.81   205.6 2274.18   215.4 2278.61
   225.2 2283.58     235 2288.64   244.8  2293.6   254.6 2298.04   264.4    2302
#Mann= 3 , 0 , 0
       0      .1       0   112.4    .045       0   127.4      .1       0
Bank Sta=112.4,127.4
XS Rating Curve= 0 ,0
Exp/Cntr=0.3,0.1

Type RM Length L Ch R = 1 ,20657.2 ,545.3,569.9,594.7
XS GIS Cut Line= 3
      1946251.44      352318.876     1946201.961      352498.564
     1946347.794      352766.793
#Sta/Elev= 30
       0 2295.78    29.4 2289.48    78.5 2279.92   107.9 2274.39   137.3 2268.59
     157 2264.92   186.4 2260.21   195.9 2259.24   205.5 2257.95   224.5 2254.51
   233.9 2253.51   243.6 2253.36   248.9 2253.61   253.2 2253.81   272.2 2255.41
   291.3  2256.7   300.9  2257.1   310.4 2257.26     320 2257.15   329.5 2257.85
     339 2260.35   348.6 2263.94   358.1 2267.84   367.6 2271.83   396.3  2284.3
   405.8 2288.17   424.9 2295.63     444 2303.44   463.1 2310.93   491.7 2322.68
#Mann= 3 , 0 , 0
       0      .1       0   233.9    .045       0   248.9      .1       0
Bank Sta=233.9,248.9
XS Rating Curve= 0 ,0
Exp/Cntr=0.3,0.1

Type RM Length L Ch R = 1 ,20087.3 ,270.3,252.9,235.2
XS GIS Cut Line= 2
     1945886.944      352193.801     1945662.898      352548.043
#Sta/Elev= 28
       0 2267.05      39  2258.8    87.7 2248.86    97.5 2246.54     117 2240.94
   126.7 2239.21   136.5 2238.47   175.5 2236.19   214.4 2234.45   224.2 2234.29
   235.7 2234.78   243.7 2235.31   253.4 2236.33   263.2 2238.68   272.9  2242.2
   282.7 2246.21   292.4 2250.29   302.2 2254.87   321.7 2264.65   331.4 2268.96
   341.2 2271.89   350.9 2274.01   360.7 2275.53   370.4 2276.66   380.2 2277.15
   389.9 2277.27   399.6 2277.18   419.2  2276.8
#Mann= 3 , 0 , 0
       0      .1       0   214.4    .045       0   235.7      .1       0
Bank Sta=214.4,235.7
XS Rating Curve= 0 ,0
Exp/Cntr=0.3,0.1

Type RM Length L Ch R = 1 ,19834.4 ,244.9,216.2,187.5
XS GIS Cut Line= 2
     1945511.857      352178.251     1945557.083      352404.305
#Sta/Elev= 27
       0 2236.86     9.6 2235.35    19.2 2234.04    28.8 2233.09    38.4 2232.59
      48 2232.36    57.6  2232.2    67.2 2232.02    76.8 2231.87    86.4 2231.76
    96.1 2231.29   105.7 2229.94   115.3 2227.88   122.1 2226.53   124.9 2225.97
   134.5 2225.21   137.1  2225.3   144.1 2225.55   153.7 2225.72   163.3 2225.88
   172.9 2227.27   182.5 2231.24   192.1 2237.14   201.7 2242.75   211.3 2246.73
   220.9 2249.23   230.5 2251.13
#Mann= 3 , 0 , 0
       0      .1       0   122.1    .045       0   144.1      .1       0
Bank Sta=122.1,144.1
XS Rating Curve= 0 ,0
Exp/Cntr=0.3,0.1

Type RM Length L Ch R = 1 ,19618.2 ,295.2,294.7,294.3
XS GIS Cut Line= 2
     1945071.753      352394.397     1945579.565      352475.126
#Sta/Elev= 30
       0 2242.19    19.4 2239.68    29.1 2238.07    67.9 2230.41      97 2223.49
   106.7 2222.11   116.4 2221.41   135.8 2220.67   164.9 2219.96   184.3 2219.92
   203.7 2220.31   223.1 2221.06   252.2 2223.02     262 2223.38   271.6 2223.23
   281.4 2222.32   300.8 2217.87   310.4 2217.05   325.4 2217.64   349.3 2219.69
   388.1 2223.68   397.8 2225.41   426.9 2233.76   436.6 2237.04   446.3 2241.01
   465.7 2249.76   475.4 2253.77   485.1 2256.85   494.8 2259.11   514.2 2263.08
#Mann= 3 , 0 , 0
       0      .1       0   300.8    .045       0   325.4      .1       0
#XS Ineff= 2 , 0
          261.13 2223.82
Permanent Ineff=
       F       F
Bank Sta=300.8,325.4
XS Rating Curve= 0 ,0
Exp/Cntr=0.3,0.1

Type RM Length L Ch R = 1 ,19323.5 ,151,150.5,149.4
XS GIS Cut Line= 2
     1944910.294      352670.439      1945501.44      352722.522
#Sta/Elev= 30
       0 2251.34    19.5 2243.89    29.2  2240.6    48.6 2235.09    77.8 2227.58
    87.6  2223.6    97.3 2217.82     107  2212.9   116.7 2210.99   126.5 2211.03
   165.4 2211.98   194.6 2212.09     214 2212.53   243.2 2212.58   262.7 2212.33
   301.6 2212.67   311.3 2212.33   326.6 2209.99   330.8  2209.3   341.6 2209.47
     360 2212.27   369.7  2212.7   447.5 2213.29   505.9  2214.5   544.8 2216.04
   554.5 2216.85   564.2 2218.65     574 2221.42   583.7 2224.73   593.4  2228.5
#Mann= 3 , 0 , 0
       0      .1       0   326.6    .045       0   341.6      .1       0
#XS Ineff= 2 , 0
          304.23 2212.99
Permanent Ineff=
       F       F
Bank Sta=326.6,341.6
XS Rating Curve= 0 ,0
Exp/Cntr=0.3,0.1

Type RM Length L Ch R = 1 ,19173   ,294.1,293.7,293.7
XS GIS Cut Line= 2
     1944941.544      352831.897     1945481.128      352857.864
#Sta/Elev= 30
       0 2222.19    19.6  2220.8    49.1 2218.55    58.9 2217.24    68.8 2213.88
    78.6 2209.12    88.4 2205.54    98.2 2204.53   117.9 2204.92   157.2    2205
   176.8 2205.18   196.4 2205.66   225.9 2206.77   235.7 2206.86   245.6  2206.2
   254.1 2205.47   255.4 2205.36   265.2 2205.12     275 2205.34   284.8 2205.51
   353.6 2206.03   432.2 2207.08     442 2207.83   451.8 2209.51   461.6 2211.51
   471.4 2213.16   481.3 2214.33   510.7 2217.24   530.4 2219.02   540.2 2220.05
#Mann= 3 , 0 , 0
       0      .1       0   254.1    .045       0     275      .1       0
#XS Ineff= 2 , 0
          234.93 2207.03
Permanent Ineff=
       F       F
Bank Sta=254.1,275
XS Rating Curve= 0 ,0
Exp/Cntr=0.3,0.1

Type RM Length L Ch R = 1 ,18879.3 ,447.5,447,446.5
XS GIS Cut Line= 2
     1944946.753      353113.147     1945429.045      353126.961
#Sta/Elev= 30
       0 2205.26      29 2205.82    38.6 2205.66    48.2 2204.74    67.6 2202.06
    77.2  2201.1    96.5 2199.66   106.2 2198.61   115.8 2197.98   135.1 2200.23
   144.8 2200.68   173.7 2200.84     193  2200.5   212.3 2199.02   231.6  2198.9
   250.9 2198.51   287.8  2197.3   299.1  2196.8   308.8 2196.89   328.1 2197.03
   337.7  2196.6   347.4  2195.8     357  2195.9   366.7  2196.8   376.3 2198.82
     386 2202.48   405.3 2211.88   443.9 2229.54   472.8 2243.18   482.5  2247.2
#Mann= 3 , 0 , 0
       0      .1       0   287.8    .045       0   308.8      .1       0
#XS Ineff= 2 , 0
          173.94 2201.17
Permanent Ineff=
       F       F
Bank Sta=287.8,308.8
XS Rating Curve= 0 ,0
Exp/Cntr=0.3,0.1

Type RM Length L Ch R = 1 ,18432.2 ,268.5,274.1,279.4
XS GIS Cut Line= 2
     1945022.273      353558.459     1945412.898      353555.855
#Sta/Elev= 30
       0  2200.7    19.5 2199.68    48.8  2196.9    58.6  2196.5    78.1 2196.52
    87.9 2195.84   107.4 2193.36   117.2 2192.49   136.7 2192.03   146.5 2191.31
   185.6 2187.66   195.3 2187.27   214.8 2187.76   224.6 2187.34   234.4 2186.04
   244.2 2185.44   253.9 2185.58   263.7 2185.24   273.4 2184.32   283.7 2183.57
     293 2183.37   298.7 2184.52   302.7 2185.32   312.5  2192.1   322.3 2202.26
     332 2211.02   341.8 2216.53   361.3 2224.32   380.9 2232.53   390.6    2236
#Mann= 3 , 0 , 0
       0      .1       0   283.7    .045       0   298.7      .1       0
Bank Sta=283.7,298.7
XS Rating Curve= 0 ,0
Exp/Cntr=0.3,0.1

Type RM Length L Ch R = 1 ,18158.2 ,318.9,321.8,327
XS GIS Cut Line= 2
      1945220.19      353803.251      1945407.69      353847.522
#Sta/Elev= 23
       0 2184.36     9.6 2184.19    19.3 2183.87    28.9 2183.49    38.5 2182.25
    48.2 2179.32    57.8 2177.26    67.4 2177.18    73.3 2176.95    77.1 2176.81
    86.7 2176.79    88.3 2177.28    96.3 2179.75     106 2185.46   115.6 2191.73
   125.2 2198.21   134.9 2205.51   144.5 2213.49   154.1 2221.62   163.8 2229.59
   173.4 2236.98     183 2243.63   192.7 2250.22
#Mann= 3 , 0 , 0
       0      .1       0    73.3    .045       0    88.3      .1       0
Bank Sta=73.3,88.3
XS Rating Curve= 0 ,0
Exp/Cntr=0.3,0.1

Type RM Length L Ch R = 1 ,17836.3 ,345.9,354.7,363.4
XS GIS Cut Line= 2
     1945074.357      354050.647     1945298.315      354180.855
#Sta/Elev= 30
       0 2183.55     9.6 2183.26    19.2 2182.09    28.8 2180.12    38.4 2177.79
      48 2175.73    57.6 2174.53    67.2 2173.79    76.8 2172.54    86.4 2170.94
    93.1 2170.68      96 2170.57   105.5 2171.27   108.1 2171.52   115.1 2172.19
   124.7 2172.81   134.3 2172.92   143.9 2172.86   153.5  2172.7   163.1 2173.23
   172.7 2176.38   182.3 2182.01   191.9  2188.8   201.5 2195.17   211.1  2200.8
   220.7 2206.71   230.3 2212.96   239.9 2219.34   249.5  2225.8   259.1 2232.35
#Mann= 3 , 0 , 0
       0      .1       0    86.4    .045       0   108.1      .1       0
Bank Sta=86.4,108.1
XS Rating Curve= 0 ,0
Exp/Cntr=0.3,0.1

Type RM Length L Ch R = 1 ,17481.7 ,419.9,430.7,441
XS GIS Cut Line= 2
     1944834.773       354227.73     1945040.503      354482.939
#Sta/Elev= 26
       0 2169.41    28.9 2167.81    57.8 2165.89    67.5 2165.33    77.1 2164.81
    86.8 2164.51    96.4 2164.44   115.7 2164.72   125.3 2164.92   163.9 2166.02
   173.5 2165.63   183.2 2163.71   187.5 2162.66   192.8 2161.37   202.5 2160.88
   212.1 2161.53   221.8 2162.61   231.4 2164.96     241 2170.95   260.3 2186.32
     270  2193.5   279.6 2200.24   289.2 2206.56   298.9 2211.99   308.5 2216.62
   327.8 2225.36
#Mann= 3 , 0 , 0
       0      .1       0   187.5    .045       0   212.1      .1       0
Bank Sta=187.5,212.1
XS Rating Curve= 0 ,0
Exp/Cntr=0.3,0.1

Type RM Length L Ch R = 1 ,17050.9 ,343.3,339.7,336.1
XS GIS Cut Line= 3
     1944527.482      354274.605     1944592.586      354613.147
     1944668.107      354753.772
#Sta/Elev= 30
       0 2158.73    19.2 2158.77    86.2 2156.95   105.3 2156.65   162.8 2156.16
   210.7 2154.95   220.2 2154.47   229.8 2153.35   239.4 2151.96     249 2151.34
   257.8 2151.96   268.1 2153.94   277.7    2156   287.3 2156.27   296.9 2154.43
   306.4 2152.87     316 2152.82   325.6 2153.35   335.2 2154.46   344.7 2157.58
   354.1  2162.6   363.5 2168.13   372.9 2173.87   391.7 2186.39   401.1 2190.97
   419.9  2197.9   429.2 2200.67     448 2205.28   457.4 2208.26   504.4 2226.19
#Mann= 3 , 0 , 0
       0      .1       0   239.4    .045       0   257.8      .1       0
#XS Ineff= 2 , 0
                          288.17         2156.62
Permanent Ineff=
       F       F
Bank Sta=239.4,257.8
XS Rating Curve= 0 ,0
Exp/Cntr=0.3,0.1

Type RM Length L Ch R = 1 ,16711.2 ,318.7,304.3,289.1
XS GIS Cut Line= 2
     1944165.503      354311.064     1944355.607      354834.501
#Sta/Elev= 30
       0 2196.84     9.8 2191.89    19.5 2186.64    39.1 2175.98    58.6 2165.08
    68.4 2160.48    78.2  2156.8    87.9 2153.57    97.7 2150.63   107.5 2148.68
   117.2 2148.35   136.8 2149.48   146.6 2149.66   185.6 2148.71   195.4 2148.15
   214.9 2145.57   224.7 2144.78   234.5 2144.78   245.9 2145.17   351.7 2148.07
   390.8 2148.72   420.1 2148.78     469  2148.1   488.5 2148.14   498.3 2149.63
     508 2153.04   517.8  2157.4   527.6 2162.39   537.4 2167.96   556.9 2180.28
#Mann= 3 , 0 , 0
       0      .1       0   224.7    .045       0   245.9      .1       0
Bank Sta=224.7,245.9
XS Rating Curve= 0 ,0
Exp/Cntr=0.3,0.1

Type RM Length L Ch R = 1 ,16406.9 ,104.3,112.8,121.3
XS GIS Cut Line= 3
     1943993.628      354649.605     1944181.128      354795.439
     1944259.253      354928.251
#Sta/Elev= 23
       0  2169.4     9.5 2165.48      19 2160.29    28.5 2153.95      38 2147.73
    47.5 2143.07      57 2140.06    66.5 2139.26      76 2139.46    78.9 2139.62
   142.5 2143.08   161.5 2143.96     171  2144.3   180.5 2144.56     190 2144.65
     209 2144.61     228 2144.37   266.4 2143.62   276.1 2145.22   285.7 2148.76
   324.2 2166.74   372.4  2188.9   391.6 2197.92
#Mann= 3 , 0 , 0
       0      .1       0      57    .045       0    78.9      .1       0
Bank Sta=57,78.9
XS Rating Curve= 0 ,0
Exp/Cntr=0.3,0.1

Type RM Length L Ch R = 1 ,16294.1 ,103.8,102.6,101.5
XS GIS Cut Line= 2
     1943936.336       354696.48     1944092.586      354951.689
#Sta/Elev= 17
       0 2165.92    38.6 2149.82    57.9 2141.97    67.6  2138.8    77.2 2137.24
    86.9 2137.06   101.9 2137.12   116.9 2137.19   135.1 2137.51   164.1 2137.71
   202.7 2137.77     222 2137.72   231.7 2138.03   241.3 2139.49     251 2142.41
   289.6 2156.18   299.2 2159.77
#Mann= 3 , 0 , 0
       0      .1       0   101.9    .045       0   116.9      .1       0
Bank Sta=101.9,116.9
XS Rating Curve= 0 ,0
Exp/Cntr=0.3,0.1

Type RM Length L Ch R = 1 ,16191.5 ,145.4,148.8,152.4
XS GIS Cut Line= 2
     1943855.694      354765.416     1944011.944      354999.791
#Sta/Elev= 22
       0 2156.43    29.1 2144.25    38.8 2140.35    48.6  2137.6    58.3 2136.59
      68 2136.63    77.7 2136.52    94.5 2135.91   106.8  2135.6   116.6 2135.89
     136 2137.32   145.7 2137.72   155.4 2137.85   165.1  2137.8   174.8 2137.63
     204 2136.66   213.7 2136.67   223.4 2137.66   233.1 2140.21   262.3 2149.76
     272 2152.98   281.7 2156.31
#Mann= 3 , 0 , 0
       0      .1       0    94.5    .045       0   116.6      .1       0
Bank Sta=94.5,116.6
XS Rating Curve= 0 ,0
Exp/Cntr=0.3,0.1

Type RM Length L Ch R = 1 ,16042.7 ,130.1,138.1,145.9
XS GIS Cut Line= 2
     1943743.628      354824.084     1943884.253      355118.355
#Sta/Elev= 25
       0 2151.98     9.6 2148.21    19.2 2144.66    38.4 2137.78      48 2134.62
    57.6 2132.35    67.2 2131.23    76.7 2130.96    95.9 2130.81   105.5 2130.51
   115.1 2130.54   124.3 2130.97   153.5 2132.29   172.7 2132.91   182.3 2133.15
   220.6 2133.63   239.8 2134.05   249.4 2134.59     259 2136.56   268.6 2140.92
   278.2 2146.17   287.8 2151.62   297.4 2157.18     307 2162.83   326.2 2174.36
#Mann= 3 , 0 , 0
       0      .1       0    95.9    .045       0   124.3      .1       0
Bank Sta=95.9,124.3
XS Rating Curve= 0 ,0
Exp/Cntr=0.3,0.1

Type RM Length L Ch R = 1 ,15904.6 ,153.7,153.8,154.4
XS GIS Cut Line= 2
     1943644.669      354844.918     1943691.544      355154.814
#Sta/Elev= 29
       0  2153.8     9.8 2149.83    19.6 2145.55    29.4 2140.84    39.2 2135.64
      49  2131.1    58.8 2128.76    68.6 2128.42    97.9 2129.04   107.7 2128.79
   117.5 2127.98   127.3 2127.65   136.5 2129.16   146.9 2130.38   156.7 2130.98
   176.3 2131.82   186.1  2132.1   195.9  2132.2   205.7 2132.15   215.5  2131.8
   225.3 2130.98   244.9 2128.78   254.6 2128.81   264.4  2131.3   274.2 2137.26
     284 2143.73   293.8  2149.9   303.6 2155.88   313.4 2161.69
#Mann= 3 , 0 , 0
       0      .1       0   117.5    .045       0   136.5      .1       0
#XS Ineff= 2 , 0
                          195.21         2132.39
Permanent Ineff=
       F       F
Bank Sta=117.5,136.5
XS Rating Curve= 0 ,0
Exp/Cntr=0.3,0.1

Type RM Length L Ch R = 1 ,15750.8 ,194.2,203.6,212.9
XS GIS Cut Line= 2
     1943511.857       354852.73     1943535.294      355170.439
#Sta/Elev= 21
       0 2151.81      29 2140.98    57.9 2130.37    67.6 2127.36    77.2 2125.83
    86.9 2125.37   106.2 2124.79   135.2 2123.49   144.8 2123.31   154.5 2123.36
   162.2  2123.6   202.7 2125.22     222  2125.9   231.7 2127.35   241.3 2130.81
     251 2135.54     280  2150.5   289.6 2155.38   299.3 2159.95   308.9 2164.23
   318.6 2168.41
#Mann= 3 , 0 , 0
       0      .1       0   135.2    .045       0   162.2      .1       0
Bank Sta=135.2,162.2
XS Rating Curve= 0 ,0
Exp/Cntr=0.3,0.1

Type RM Length L Ch R = 1 ,15547.2 ,152.6,159.9,167.2
XS GIS Cut Line= 2
     1943371.232      354826.689     1943257.921      355152.037
#Sta/Elev= 29
       0 2150.52     9.6 2147.49    19.1 2144.33    28.7 2140.95    57.4 2130.48
      67 2127.11    76.6 2124.42    86.1 2122.92   114.8 2120.88   124.4 2120.61
     134 2120.92   137.1  2121.1   153.1 2121.95   162.7 2122.33   191.4 2123.16
   210.5 2123.27   229.7 2123.02   239.2 2123.63   248.8 2126.28   258.4 2131.26
     268 2136.93   277.5 2141.94   287.1    2146   296.7 2149.64   306.2 2152.82
   315.8 2154.63   325.4 2154.24     335 2152.38   344.5 2150.22
#Mann= 3 , 0 , 0
       0      .1       0   114.8    .045       0   137.1      .1       0
Bank Sta=114.8,137.1
XS Rating Curve= 0 ,0
Exp/Cntr=0.3,0.1

Type RM Length L Ch R = 1 ,15387.3 ,108.7,109.7,110.7
XS GIS Cut Line= 2
     1943252.395      354800.138     1943096.453      355004.311
#Sta/Elev= 30
       0 2136.65     9.5 2134.28      19 2131.97    28.6 2129.67    38.1 2127.33
    47.6 2124.84    57.1 2122.23    66.6 2119.87    76.1 2118.55    85.6 2118.01
    95.2  2117.4   104.7 2116.51   105.3 2116.45   114.2  2115.5   120.3 2115.28
   123.7 2115.15   133.2 2115.57   142.7 2115.73   152.2 2115.64   161.8 2115.98
   171.3 2118.27   180.8 2121.77   190.3 2125.58   199.8 2129.17   209.3 2132.38
   218.8 2135.34   228.4 2137.99   237.9 2138.71   247.4 2137.61   256.9 2135.93
#Mann= 3 , 0 , 0
       0      .1       0   105.3    .045       0   133.2      .1       0
Bank Sta=105.3,133.2
XS Rating Curve= 0 ,0
Exp/Cntr=0.3,0.1

Type RM Length L Ch R = 1 ,15277.6 ,204,177.5,151.1
XS GIS Cut Line= 2
     1943219.843       354676.44     1943028.871      354906.475
#Sta/Elev= 30
       0 2170.57     9.6 2166.92    19.3 2162.82    28.9 2158.43    38.6 2153.37
    48.2 2147.96    57.9 2142.05    67.5 2137.18    77.2 2133.22    86.8 2129.89
    96.4 2126.94   106.1 2124.15   125.4 2118.41     135 2116.26   144.7 2115.41
     164 2114.93   173.6 2114.56   183.2 2114.04   192.9 2113.31   202.5 2112.48
   212.2 2112.16   221.8 2112.56   231.5 2113.26   241.1 2115.03   250.8 2117.84
   260.4 2121.01     270 2124.05   279.7 2127.01   289.3 2128.58     299 2127.76
#Mann= 3 , 0 , 0
       0      .1       0   192.9    .045       0   221.8      .1       0
Bank Sta=192.9,221.8
XS Rating Curve= 0 ,0
Exp/Cntr=0.3,0.1

Type RM Length L Ch R = 1 ,15100   ,240.3,214.3,188.2
XS GIS Cut Line= 2
     1942811.857      354552.742     1942991.979      354956.388
#Sta/Elev= 30
       0 2162.27     9.8  2155.4    19.6 2149.27    29.5 2143.38    39.3 2137.78
    49.1 2133.16    58.9 2129.24    68.8 2126.01    78.6 2123.18    88.4 2120.66
    98.2  2118.4     108 2116.37   117.9 2114.45   127.7 2112.72   137.5  2111.4
   147.3 2110.73   186.6 2110.02   245.6  2109.3     275 2108.13   294.7 2106.94
   304.5 2106.42   314.3 2106.51   324.1 2107.19     334 2108.18   353.6 2110.59
   363.4 2111.66   392.9 2114.41   412.5  2116.4   422.4 2117.46     442 2119.75
#Mann= 3 , 0 , 0
       0      .1       0   294.7    .045       0   324.1      .1       0
Bank Sta=294.7,324.1
XS Rating Curve= 0 ,0
Exp/Cntr=0.3,0.1

Type RM Length L Ch R = 1 ,14885.7 ,338.6,329.6,320
XS GIS Cut Line= 2
     1942459.773      354988.147     1943014.461      354998.564
#Sta/Elev= 30
       0 2183.58     9.7 2185.98    19.5 2187.93    48.7 2191.31    68.1 2194.18
   126.5 2205.54   136.3 2207.07     146 2205.89   155.7 2199.52   165.5 2189.24
   175.2 2177.87   184.9  2166.1   194.7 2153.03   214.1 2123.46   223.9 2111.01
   233.6 2103.91   243.3 2101.89   330.9 2101.24   379.6  2101.6   399.1 2101.08
     403  2101.1     418 2101.56   428.3 2103.38     438 2106.99   447.7 2109.49
   457.4 2110.52   496.4 2111.72   506.1 2112.77   525.6 2115.96   554.8 2122.17
#Mann= 3 , 0 , 0
       0      .1       0     403    .045       0     418      .1       0
Bank Sta=403,418
XS Rating Curve= 0 ,0
Exp/Cntr=0.3,0.1

Type RM Length L Ch R = 1 ,14556.1 ,328.2,337,346.1
XS GIS Cut Line= 2
     1942783.613      355359.673     1943224.586      355172.173
#Sta/Elev= 30
       0 2105.73    19.6 2110.72    29.3 2114.01    48.9 2121.94    68.4  2130.6
    78.2 2133.98      88 2136.38    97.8 2137.46   107.6 2136.94   117.4 2135.18
   136.9 2128.42   166.2 2115.47   195.6 2101.38   205.4 2097.33   215.1 2093.98
   234.7 2091.28   244.5 2089.48   254.3 2086.85     264 2085.11   273.8 2084.61
   293.4 2084.98   322.7 2087.31   332.5 2089.62   342.3 2094.28     352 2099.84
   361.8 2104.57   381.4 2111.89   430.3 2128.09   449.8 2133.22   479.2 2139.81
#Mann= 3 , 0 , 0
       0      .1       0   254.3    .045       0   273.8      .1       0
Bank Sta=254.3,273.8
XS Rating Curve= 0 ,0
Exp/Cntr=0.3,0.1

Type RM Length L Ch R = 1 ,14219.1 ,311.8,342.8,373.6
XS GIS Cut Line= 3
     1942882.572      355364.447     1942983.483      355562.053
     1943462.161      355563.451
#Sta/Elev= 30
       0 2123.87    19.3 2118.63    38.6 2114.76    57.9 2111.76    77.2 2109.58
   135.1 2099.47   183.3 2086.69   202.6 2083.84   221.9 2081.75   270.7  2081.5
   290.3 2079.39     300  2079.4   348.9 2081.13   358.6 2080.99   368.4 2080.16
   378.2 2079.02     388  2079.5  391.54 2080.89   397.7  2083.4   407.5 2089.21
   417.3 2094.32     427 2097.96   446.6 2101.82   485.6 2111.47   505.2 2114.67
   544.3 2119.76     554 2121.49   583.3  2127.9   632.2 2133.97   700.6 2143.52
#Mann= 3 , 0 , 0
       0      .1       0   368.4    .045       0  391.54      .1       0
Bank Sta=368.4,391.54
XS Rating Curve= 0 ,0
Exp/Cntr=0.3,0.1

Type RM Length L Ch R = 1 ,13876.3 ,181.3,194.5,207.8
XS GIS Cut Line= 2
     1942950.659       355573.65     1943072.187      356129.206
#Sta/Elev= 30
       0 2079.49    19.6 2076.98    29.4 2075.98    39.2 2075.31      49 2074.97
    78.4 2074.73   117.7 2075.02   166.7 2074.46   205.9 2074.55   235.3 2074.24
   264.7 2073.05   274.5  2072.1   283.9 2070.79   294.2 2069.64     304 2069.96
   313.8 2072.82   323.6 2079.15   343.2 2096.34     353 2104.62   362.8 2112.43
   382.4 2127.27   392.2 2133.77     402  2138.5   411.8 2142.53   431.4 2151.07
   460.8 2163.52   480.4 2172.19   500.1 2179.62   519.7 2186.67   568.7 2204.73
#Mann= 3 , 0 , 0
       0      .1       0   283.9    .045       0     304      .1       0
Bank Sta=283.9,304
XS Rating Curve= 0 ,0
Exp/Cntr=0.3,0.1

Type RM Length L Ch R = 1 ,13681.8 ,259.8,274.2,288.5
XS GIS Cut Line= 2
     1942936.625      355514.478     1942797.736      355894.686
#Sta/Elev= 28
       0  2092.2    19.3 2087.62    28.9 2085.62    48.2  2081.9    57.8 2079.82
    77.1 2074.92    86.7 2072.98    96.4 2072.11     106 2071.95   115.6  2071.9
   163.8 2070.69   250.6 2069.05   269.8 2068.57   279.5  2068.1   289.1 2067.01
   298.8 2065.02   308.4 2063.89     318 2064.03   322.6 2065.66   327.7 2067.47
   337.3 2076.44     347 2088.59   356.6 2099.75   366.2 2108.39   375.9 2115.58
   385.5 2122.47   395.1 2128.92   404.8 2134.24
#Mann= 3 , 0 , 0
       0      .1       0   298.8    .045       0   322.6      .1       0
Bank Sta=298.8,322.6
XS Rating Curve= 0 ,0
Exp/Cntr=0.3,0.1

Type RM Length L Ch R = 1 ,13407.6 ,237.2,231.4,225.8
XS GIS Cut Line= 2
     1942804.681      355516.214     1942587.667      355660.311
#Sta/Elev= 30
       0 2078.38     9.6 2077.33    19.3 2075.96    28.9 2074.15    38.6 2071.98
    48.2  2069.7    57.9 2067.56    67.5 2065.94    77.2 2064.79    86.8 2063.84
    96.5    2063   106.1 2062.26   115.8 2061.69   125.4 2061.27   135.1 2060.51
   144.7 2059.01   154.4  2057.3     164 2056.22   173.7 2056.23   176.4 2056.23
   183.3 2056.22   191.4 2057.65     193 2057.93   202.6  2061.8   212.3 2066.88
   221.9 2071.88   231.6  2076.3   241.2 2080.51   250.8 2084.69   260.5 2089.08
#Mann= 3 , 0 , 0
       0      .1       0   154.4    .045       0   191.4      .1       0
Bank Sta=154.4,191.4
XS Rating Curve= 0 ,0
Exp/Cntr=0.3,0.1

Type RM Length L Ch R = 1 ,13176.2 ,156.9,142.6,128
XS GIS Cut Line= 2
     1942660.584      355278.367     1942462.667      355511.006
#Sta/Elev= 30
       0 2113.05     9.5 2108.31    19.1 2103.36    38.2 2093.03    47.7 2087.81
    57.3  2082.7    66.8 2077.92    76.4 2073.69    85.9 2070.11    95.4 2066.72
     105 2063.12   114.5 2059.33   124.1 2056.01   133.6 2054.62   152.7 2053.53
   162.3 2052.12   171.8 2050.57   181.4 2050.04   185.4 2050.07   200.4 2050.22
     210 2050.29   229.1 2050.64   238.6 2051.03   248.2 2052.18   257.7 2054.91
   267.3 2058.64   276.8 2061.72   286.4 2063.34   295.9 2064.18   305.4 2064.78
#Mann= 3 , 0 , 0
       0      .1       0   185.4    .045       0   200.4      .1       0
Bank Sta=185.4,200.4
XS Rating Curve= 0 ,0
Exp/Cntr=0.3,0.1

Type RM Length L Ch R = 1 ,13033.6 ,267.5,258.8,250.1
XS GIS Cut Line= 2
     1942408.847      355262.742     1942388.014      355493.645
#Sta/Elev= 27
       0 2061.15     9.7 2058.58    19.3 2055.95      29 2053.43    38.6 2051.61
    48.3 2050.94      58 2050.98    67.6 2051.22    77.3 2051.51    86.9 2051.63
    96.6 2051.23   106.3 2049.87   115.9 2047.58   125.6 2045.45   133.1 2044.76
   135.2 2044.57   144.9 2045.14   148.1 2045.67   154.6 2046.74   164.2 2048.72
   173.9 2051.21   183.5 2054.74   193.2 2058.71   202.9 2061.97   212.5 2063.97
   222.2 2065.16   231.8 2066.19
#Mann= 3 , 0 , 0
       0      .1       0   125.6    .045       0   148.1      .1       0
Bank Sta=125.6,148.1
XS Rating Curve= 0 ,0
Exp/Cntr=0.3,0.1

Type RM Length L Ch R = 1 ,12774.8 ,209,206.7,204.4
XS GIS Cut Line= 2
     1942105.028      355297.464     1942158.847      355476.284
#Sta/Elev= 22
       0 2061.33     9.8 2052.01    19.7 2043.92    29.5 2040.73    39.3 2040.46
    49.1 2040.28      59 2040.15    68.8 2040.07    78.6 2039.93    88.5 2039.52
    98.3 2038.75   108.1 2037.99   110.3 2037.93   117.9 2037.72   125.3 2037.93
   127.8    2038   137.6 2038.74   147.4 2039.68   157.3    2041   167.1 2042.82
   176.9 2044.96   186.7 2047.22
#Mann= 3 , 0 , 0
       0      .1       0   110.3    .045       0   125.3      .1       0
Bank Sta=110.3,125.3
XS Rating Curve= 0 ,0
Exp/Cntr=0.3,0.1

Type RM Length L Ch R = 1 ,12568.1 ,487.3,485.7,484
XS GIS Cut Line= 2
     1941914.056      355398.159     1941985.236      355573.506
#Sta/Elev= 23
       0 2050.57     9.5  2047.3    18.9  2043.7    28.4 2039.44    37.8 2035.17
    47.3 2032.07    56.1 2031.21    56.8 2031.14    66.2 2031.14    71.1 2031.32
    75.7 2031.48    85.2  2031.9    94.6 2032.33   104.1 2032.73   113.6 2033.22
     123 2034.33   132.5 2036.86   141.9 2040.29   151.4 2043.65   160.9 2046.99
   170.3 2050.19   179.8 2052.94   189.2  2055.2
#Mann= 3 , 0 , 0
       0      .1       0    56.1    .045       0    71.1      .1       0
Bank Sta=56.1,71.1
XS Rating Curve= 0 ,0
Exp/Cntr=0.3,0.1

Type RM Length L Ch R = 1 ,12082.4 ,206,216.4,226.7
XS GIS Cut Line= 2
     1941469.611      355498.853     1941544.264      355656.839
#Sta/Elev= 21
       0 2024.86     9.7 2023.94    19.4 2022.88    29.1 2020.95    38.8 2018.01
    42.5 2017.08    48.5 2015.56    57.5 2014.87    58.2 2014.82      68 2014.78
    77.7 2014.74    87.4 2015.64    97.1 2017.75   106.8  2019.3   116.5 2020.11
   126.2 2020.82   135.9 2021.58   145.6 2022.42   155.3 2024.17     165 2027.34
   174.7  2031.2
#Mann= 3 , 0 , 0
       0      .1       0    48.5    .045       0    87.4      .1       0
Bank Sta=48.5,87.4
XS Rating Curve= 0 ,0
Exp/Cntr=0.3,0.1

Type RM Length L Ch R = 1 ,11866   ,163,162.3,161.5
XS GIS Cut Line= 3
     1941328.986      355377.325     1941294.264       355478.02
     1941290.792      355668.992
#Sta/Elev= 24
       0 2062.32     9.7 2057.58      29 2047.98    38.7 2043.59    48.4 2039.48
    58.1 2036.02    77.5 2030.49    87.2 2027.38    96.8 2023.81   106.5 2020.78
   116.1 2018.98   125.6 2018.06   173.4 2014.23   182.9 2013.62     202 2012.63
   211.6 2011.47   216.4 2010.48   221.1 2009.52   230.7 2008.05   240.2 2008.08
   249.8 2009.64   259.3 2013.07     288 2025.87   297.5  2030.2
#Mann= 3 , 0 , 0
       0      .1       0   216.4    .045       0   249.8      .1       0
Bank Sta=216.4,249.8
XS Rating Curve= 0 ,0
Exp/Cntr=0.3,0.1

Type RM Length L Ch R = 1 ,11703.7 ,178.2,197.2,216.5
XS GIS Cut Line= 2
     1941127.597      355359.964     1941134.976      355684.183
#Sta/Elev= 24
       0 2046.39     9.8 2041.92    19.6 2037.61    29.5 2033.67    68.8 2018.62
    78.6 2015.26    88.4 2013.04    98.3 2012.22   117.9 2011.86   157.2 2011.52
   196.6  2011.7   206.4 2011.17   216.2 2009.37   221.1 2008.11     226 2006.85
   235.9 2005.83   245.7 2006.47   265.3 2008.56   275.2 2011.25     285  2016.3
   294.8 2022.58   304.6 2029.02   314.5 2035.04   324.3 2040.38
#Mann= 3 , 0 , 0
       0      .1       0   221.1    .045       0   245.7      .1       0
Bank Sta=221.1,245.7
XS Rating Curve= 0 ,0
Exp/Cntr=0.3,0.1

Type RM Length L Ch R = 1 ,11506.5 ,286.1,266.1,245.1
XS GIS Cut Line= 2
     1941054.681      355456.318      1940887.58      355614.738
#Sta/Elev= 27
       0 2009.53     9.6 2008.78    19.2 2008.01    28.8 2007.26    38.4 2006.62
      48  2006.2    57.6 2005.97    67.2 2006.02    76.8 2006.52    86.4 2007.04
    95.9 2007.35   105.5 2006.74   115.1 2005.25   124.7  2003.4   134.3 2001.32
   139.4 2000.51   143.9  1999.8   153.5 1999.54   154.4 1999.64   163.1 2000.62
   172.7 2004.24   182.3 2009.44   191.9 2015.21   201.5 2020.52   211.1 2024.15
   220.7 2026.65   230.3 2028.71
#Mann= 3 , 0 , 0
       0      .1       0   139.4    .045       0   163.1      .1       0
Bank Sta=139.4,163.1
XS Rating Curve= 0 ,0
Exp/Cntr=0.3,0.1

Type RM Length L Ch R = 1 ,11240.4 ,272.5,269.9,267.1
XS GIS Cut Line= 3
     1940761.712      355356.492     1940718.309      355464.999
     1940720.479      355586.527
#Sta/Elev= 28
       0 2061.47     9.7 2056.92    19.5 2052.03    29.2  2046.9      39 2041.83
    48.7 2036.78    58.4 2031.85    68.2 2026.86    77.9 2021.77    87.6 2016.63
    97.4 2011.56   107.1 2006.77   116.9 2002.26   126.2  1998.1   135.6 1994.02
   142.3  1992.2   144.9  1991.5   154.3 1991.16   157.3 1991.71   163.6 1992.86
     173  1995.4   182.3 1997.81   191.7 1999.98     201 2002.34   210.4 2004.83
   219.7 2007.42   229.1 2010.15   238.4 2013.15
#Mann= 3 , 0 , 0
       0      .1       0   142.3    .045       0   157.3      .1       0
Bank Sta=142.3,157.3
XS Rating Curve= 0 ,0
Exp/Cntr=0.3,0.1

Type RM Length L Ch R = 1 ,10970.5 ,294.9,294.4,293.7
XS GIS Cut Line= 2
     1940440.531      355378.193     1940494.785      355697.204
#Sta/Elev= 30
       0 2025.99     9.8 2023.94    19.6 2022.32    29.4 2021.22    39.2 2020.48
    58.8 2019.35    68.6 2018.65    78.4 2017.64    88.2 2016.26    98.1 2014.69
   107.9 2013.26   137.3 2009.61   147.1 2008.08   156.9 2005.98   166.7 2003.18
   176.5 1999.78   186.3 1995.93   196.1  1991.7   201.9 1989.41   205.9 1987.83
   215.7 1986.04   225.5 1987.58   235.3 1992.66   245.1  1999.3     255 2005.31
   284.4 2022.62   294.2 2028.01     304 2032.44   313.8 2035.83   323.6    2039
#Mann= 3 , 0 , 0
       0      .1       0   201.9    .045       0   225.5      .1       0
Bank Sta=201.9,225.5
XS Rating Curve= 0 ,0
Exp/Cntr=0.3,0.1

Type RM Length L Ch R = 1 ,10676.1 ,249.3,267.8,286.3
XS GIS Cut Line= 2
     1940173.733      355475.594      1940221.22      355704.398
#Sta/Elev= 27
       0  2006.9     9.7 2005.25    19.5  2000.9    29.2 1994.25      39 1987.66
    48.7 1982.72    58.4 1978.64    68.2 1974.21      76 1971.64    77.9 1971.02
    87.6  1971.1      91  1972.4    97.4 1974.85   107.1 1979.42   116.8 1983.04
   126.6 1986.04   136.3 1988.42     146 1989.86   155.8 1990.95   165.5  1992.1
   175.3 1993.35     185 1994.64   194.7  1995.9   204.5 1997.23   214.2 1999.08
   223.9 2002.06   233.7 2005.78
#Mann= 3 , 0 , 0
       0      .1       0      76    .045       0      91      .1       0
Bank Sta=76,91
XS Rating Curve= 0 ,0
Exp/Cntr=0.3,0.1

Type RM Length L Ch R = 1 ,10408.3 ,98.4,106.5,114.4
XS GIS Cut Line= 2
     1940024.107      355434.136     1939862.904      355669.862
#Sta/Elev= 28
       0 2007.03     9.5 2006.11      19 2004.17    28.6 2001.08    38.1 1997.37
    47.6 1993.45    57.1 1989.69    85.7 1975.46    95.2 1970.97   114.2 1962.49
   123.8 1958.36   133.3  1955.4   142.8 1953.62   152.3 1952.24   156.2  1951.6
   161.8 1950.67   171.2  1950.1   180.9 1949.93   190.4  1949.5   199.9 1948.58
   209.4 1948.09   218.9 1950.15   228.5 1955.02     238 1961.47   247.5 1967.38
     257 1969.83   266.5 1970.76   285.6 1971.32
#Mann= 3 , 0 , 0
       0      .1       0   156.2    .045       0   171.2      .1       0
Bank Sta=156.2,171.2
XS Rating Curve= 0 ,0
Exp/Cntr=0.3,0.1

Type RM Length L Ch R = 1 ,10301.8 ,193.7,165.7,137.2
XS GIS Cut Line= 3
     1939956.139      355427.381     1939813.995      355527.207
     1939823.761      355674.777
#Sta/Elev= 25
       0 1980.01     9.6 1976.24      29 1969.07    38.6 1965.44    57.9 1957.62
    67.6 1953.82    77.2  1950.6    86.8 1948.53   106.2 1945.14   115.8 1943.25
   125.4 1941.69   135.1 1941.26   154.4 1941.29   173.7 1941.31   201.4 1942.13
   219.9 1942.44   229.2  1942.8   238.4  1944.1   247.6 1947.02   256.9  1951.2
   275.4 1960.32   284.6 1963.99   293.9 1965.91   303.1 1966.84   321.6 1968.34
#Mann= 3 , 0 , 0
       0      .1       0   125.4    .045       0   154.4      .1       0
Bank Sta=125.4,154.4
XS Rating Curve= 0 ,0
Exp/Cntr=0.3,0.1

Type RM Length L Ch R = 1 ,10136.1 ,277.1,254.3,231.4
XS GIS Cut Line= 2
      1939707.49      355302.912     1939776.563      355622.374
#Sta/Elev= 29
       0 2005.41     9.6    1998    19.2 1991.06    38.4 1977.83    48.1 1970.99
    57.7 1963.57    67.3  1955.3    76.9 1946.35    86.5  1938.2    96.1 1932.77
   105.7 1930.12   115.4 1928.94     125 1928.74   135.6 1929.74   144.2 1930.82
   153.8 1931.89     173 1933.66   201.9 1936.74   211.5 1937.55   221.1 1938.03
   240.3 1938.53   249.9 1938.61   269.2 1938.58   278.8 1938.64   288.4 1938.98
     298 1940.27   307.6  1943.1   317.2 1947.13   326.8 1951.57
#Mann= 3 , 0 , 0
       0      .1       0   115.4    .045       0   135.6      .1       0
Bank Sta=115.4,135.6
XS Rating Curve= 0 ,0
Exp/Cntr=0.3,0.1

Type RM Length L Ch R = 1 ,9881.9  ,344.6,376.8,409.1
XS GIS Cut Line= 3
     1939448.466      355536.033       1939634.1      355605.106
     1939685.905      355808.008
#Sta/Elev= 30
       0  1930.9    18.9 1930.24    28.3 1929.53    37.7 1928.44    47.2 1926.68
    56.6 1923.44      66 1918.81   71.831917.018    75.4 1915.92    84.9 1915.92
    94.3 1917.23     102 1918.72     132 1924.12   160.3 1930.02   169.8  1931.8
   179.2 1933.03   198.1 1934.78   207.6 1935.98   217.1 1937.26   226.6 1939.03
   236.1 1941.54   264.7 1950.73   274.2 1953.49   283.7  1955.6   312.3  1960.9
   321.8 1962.92   331.3 1965.22   369.4 1975.12   378.9  1977.7   407.5 1986.25
#Mann= 3 , 0 , 0
       0      .1       0   71.83    .045       0     102      .1       0
Bank Sta=71.83,102
XS Rating Curve= 0 ,0
Exp/Cntr=0.3,0.1

Type RM Length L Ch R = 1 ,9505    ,212.9,204.9,197
XS GIS Cut Line= 2
     1939249.881      355484.228     1939198.077       355760.52
#Sta/Elev= 26
       0 1911.75    19.4 1909.87    29.1 1908.83    38.8  1907.7    48.5 1906.44
    87.2 1901.14    96.9  1899.5   106.6 1897.74   116.3  1896.7     126 1896.92
   138.4 1897.77   145.4 1898.13   155.1 1898.48   164.8 1899.44   174.5 1902.36
   184.2 1907.44   193.9  1913.5   203.6 1919.68   213.2 1925.21     223 1928.96
   232.6  1930.8   242.3 1931.73     252 1932.42   261.7 1932.96   271.4 1933.36
   281.1 1933.65
#Mann= 3 , 0 , 0
       0      .1       0   106.6    .045       0   138.4      .1       0
Bank Sta=106.6,138.4
XS Rating Curve= 0 ,0
Exp/Cntr=0.3,0.1

Type RM Length L Ch R = 1 ,9300.1  ,282.4,288,292.8
XS GIS Cut Line= 2
     1939012.443      355492.862     1939051.297      355721.667
#Sta/Elev= 26
       0 1914.13     9.7 1911.43    19.3  1908.8      29 1906.22    38.7 1903.66
    48.4  1901.1      58 1898.35    67.7 1894.78    77.4  1891.5      87 1890.32
    91.2 1890.63    96.7 1891.04   106.2 1892.04     116 1893.71   125.7 1896.02
   135.4 1897.92     145 1899.29   154.7 1900.39   164.4 1901.51   174.1 1902.76
   183.7 1904.12   193.4 1905.43   203.1 1906.57   212.7 1907.69   222.4 1908.88
   232.1 1910.11
#Mann= 3 , 0 , 0
       0      .1       0    77.4    .045       0   106.2      .1       0
Bank Sta=77.4,106.2
XS Rating Curve= 0 ,0
Exp/Cntr=0.3,0.1

Type RM Length L Ch R = 1 ,9012.1  ,348.1,350.4,352.5
XS GIS Cut Line= 2
     1938755.868      355544.496     1938742.847       355765.85
#Sta/Elev= 26
       0 1893.24     9.6  1890.6    19.3 1887.97    28.9 1885.51    38.6 1883.65
    48.2 1882.54    57.8 1881.82    67.5 1881.11    77.1 1880.18    86.8 1878.92
    91.5 1878.14    96.4 1877.33     106 1875.88   106.5 1875.86   115.7 1875.53
   125.3 1877.78     135 1880.89   144.6 1883.48   154.2 1885.67   163.9 1887.75
   173.5 1889.69   183.2 1891.54   192.8 1893.16   202.5 1895.09   212.1 1897.71
   221.7 1900.35
#Mann= 3 , 0 , 0
       0      .1       0    91.5    .045       0   125.3      .1       0
Bank Sta=91.5,125.3
XS Rating Curve= 0 ,0
Exp/Cntr=0.3,0.1

Type RM Length L Ch R = 1 ,8661.7  ,257,250.7,244.4
XS GIS Cut Line= 4
     1938447.708      355498.923     1938408.645      355585.728
     1938397.686      355654.463     1938410.816      355741.978
#Sta/Elev= 30
       0 1869.23     9.5  1866.5      19 1863.64    28.6 1860.71    38.1 1857.72
    47.6 1854.65    57.1 1851.61    66.6 1848.56    76.2 1845.58    85.7 1842.79
    95.2 1840.27   103.9 1838.32   112.6 1836.45   117.1 1835.59   121.3 1834.78
     130 1833.86   132.1 1833.92   138.7  1834.1   147.4 1835.67   156.1 1837.89
   164.8 1840.04   174.6 1842.41   184.5 1844.76   194.3 1847.18   204.1 1849.57
     214 1851.92   223.8 1854.33   233.6 1857.24   243.4    1861   253.3 1865.27
#Mann= 3 , 0 , 0
       0      .1       0   117.1    .045       0   147.4      .1       0
Bank Sta=117.1,147.4
XS Rating Curve= 0 ,0
Exp/Cntr=0.3,0.1

Type RM Length L Ch R = 1 ,8411    ,206.4,204.5,202.6
XS GIS Cut Line= 4
     1938187.291      355477.221     1938153.858       355551.11
     1938167.886      355670.349     1938208.993      355720.277
#Sta/Elev= 22
       0 1844.83      27 1837.85    45.1 1833.08    54.1 1830.62    63.1 1828.02
    72.1 1825.06    81.1  1821.8    90.3 1817.58    99.6 1813.84   108.8 1813.48
     118 1814.57   127.3 1815.75   136.5 1816.53     155 1817.56   173.5 1818.69
   191.9 1820.05   201.2 1820.82   228.9 1825.02   238.1 1826.66   247.4 1829.12
   256.6 1832.95   265.8 1837.37
#Mann= 3 , 0 , 0
       0      .1       0    99.6    .045       0     118      .1       0
Bank Sta=99.6,118
XS Rating Curve= 0 ,0
Exp/Cntr=0.3,0.1

Type RM Length L Ch R = 1 ,8206.5  ,448.1,453.7,459.2
XS GIS Cut Line= 4
     1938006.568      355505.814     1937950.446      355583.521
     1937980.665      355730.301     1938067.007      355803.691
#Sta/Elev= 29
       0 1815.12    19.2 1810.42    38.3 1805.56    67.1 1797.81    76.7 1795.28
    95.8  1790.4   105.2 1788.85   114.6 1787.46     124 1786.41   133.3 1785.58
   143.5 1784.45     152  1783.3   161.4 1782.52   170.8 1783.06   189.5 1786.43
   198.9 1787.85   217.6 1790.26     227 1791.37   245.7 1793.28   255.2 1795.18
   264.6 1797.38     274 1800.97   283.5 1806.28   292.9 1811.94   302.4 1816.95
   311.8 1821.17   321.3  1825.6   340.1 1835.29     359 1844.88
#Mann= 3 , 0 , 0
       0      .1       0   143.5    .045       0   170.8      .1       0
Bank Sta=143.5,170.8
XS Rating Curve= 0 ,0
Exp/Cntr=0.3,0.1

Type RM Length L Ch R = 1 ,7752.9  ,597,581.8,566.5
XS GIS Cut Line= 2
     1937522.219       355447.05     1937505.789      355829.593
#Sta/Elev= 30
       0 1760.03    19.6  1753.5    49.1 1745.56    58.9 1743.39    68.7 1741.85
    98.2 1738.74     108 1737.28   117.8 1735.27   127.6 1732.59   157.1  1723.9
   166.9 1720.47   186.5 1712.46   196.4 1707.92   206.2 1702.85     216 1698.64
   217.1 1698.45   225.8 1696.95   235.6 1697.92   245.4 1700.44   265.1  1706.8
   274.9  1710.9   284.7  1715.6   294.5 1720.85   304.4 1726.77   314.2 1733.71
     324    1742   343.6 1760.61   353.4 1768.49   363.3 1774.11   382.9 1782.09
#Mann= 3 , 0 , 0
       0      .1       0   217.1    .045       0   235.6      .1       0
Bank Sta=217.1,235.6
XS Rating Curve= 0 ,0
Exp/Cntr=0.3,0.1

Type RM Length L Ch R = 1 ,7171.1  ,490.8,494.5,498.1
XS GIS Cut Line= 2
     1936888.449      355536.033     1937052.497       355760.52
#Sta/Elev= 22
       0 1682.37    19.2 1672.49    28.8 1667.92    38.4 1663.73    47.9 1660.01
    57.5 1656.63    67.1 1653.59    76.7 1650.88    86.3 1648.33    95.9 1645.56
   113.5 1639.59     115 1639.08   124.6 1637.58   134.2 1639.03   143.8 1642.06
   153.4 1645.31   172.6 1650.38   182.2 1653.07   191.8 1656.19   220.5 1666.63
   249.3 1676.76     278 1687.28
#Mann= 3 , 0 , 0
       0      .1       0   113.5    .045       0   134.2      .1       0
Bank Sta=113.5,134.2
XS Rating Curve= 0 ,0
Exp/Cntr=0.3,0.1

Type RM Length L Ch R = 1 ,6676.5  ,571.5,575.1,577.9
XS GIS Cut Line= 2
     1936486.962      355777.788      1936607.84      356019.544
#Sta/Elev= 18
       0 1618.22     9.6 1614.88    48.3 1601.87    57.9  1598.9    67.6 1596.32
    77.2 1593.95    86.9 1591.21    96.5  1588.1   106.2 1585.92   125.5 1585.25
   144.8 1583.69   154.4  1583.5   164.1 1585.63   173.8 1589.74   212.4 1607.04
   241.3 1620.32   260.6 1628.52   270.3 1632.54
#Mann= 3 , 0 , 0
       0      .1       0   125.5    .045       0   164.1      .1       0
Bank Sta=125.5,164.1
XS Rating Curve= 0 ,0
Exp/Cntr=0.3,0.1

Type RM Length L Ch R = 1 ,6101.5  ,399.3,404.4,409.5
XS GIS Cut Line= 2
     1935973.232      355972.056     1936050.939      356200.861
#Sta/Elev= 28
       0 1566.84     9.7 1564.84    19.3  1562.1      29 1558.79    38.7 1555.43
    48.3 1552.04      58 1548.66    67.7 1545.35    77.3 1542.08      87 1538.86
    96.7 1535.67   106.3 1532.22     116 1528.08   125.6 1524.29   130.7 1523.86
   135.3 1523.48     145 1526.74   145.7 1527.06   154.6 1531.08   164.3 1534.69
     174 1537.68   183.6 1540.72   193.3 1543.88     203 1547.12   212.6 1550.46
   222.3 1553.88     232 1557.33   241.6 1560.82
#Mann= 3 , 0 , 0
       0      .1       0   125.6    .045       0   145.7      .1       0
Bank Sta=125.6,145.7
XS Rating Curve= 0 ,0
Exp/Cntr=0.3,0.1

Type RM Length L Ch R = 1 ,5697.1  ,381.1,385.3,389.3
XS GIS Cut Line= 2
     1935619.233      356071.349     1935645.135      356321.738
#Sta/Elev= 29
       0 1521.73     9.7 1520.04    19.4 1517.56      29 1515.99    38.7  1513.9
    48.4 1509.66    58.1  1504.7    67.8 1500.04    77.4 1496.42    87.1  1494.1
    96.8 1492.39   106.5 1490.75   107.8  1490.6   116.2 1489.62   122.8 1489.65
   125.9 1489.66   135.5 1490.84   145.2 1492.44   154.9 1493.91   164.6 1495.79
   174.3 1499.29     184 1504.41   193.6 1509.74   203.3 1513.58     213 1514.74
   222.7 1514.41   232.4 1515.64     242 1519.32   251.7 1523.71
#Mann= 3 , 0 , 0
       0      .1       0   107.8    .045       0   135.5      .1       0
Bank Sta=107.8,135.5
XS Rating Curve= 0 ,0
Exp/Cntr=0.3,0.1

Type RM Length L Ch R = 1 ,5311.8  ,206.7,209.2,211.4
XS GIS Cut Line= 2
     1935259.774      356126.093     1935248.923      356327.916
#Sta/Elev= 24
       0 1471.87     9.6 1469.49    19.2 1468.32    28.9 1468.21    38.5    1468
    48.1 1467.05    57.8 1465.84    67.4 1464.88      77 1464.28    83.5 1463.97
    86.6 1463.82    96.2 1463.46    98.5 1463.58   105.9 1463.96   115.5 1465.04
   125.1 1465.86   134.7 1466.45   144.4 1467.87     154 1470.72   163.6 1474.65
   173.2 1479.69   182.9 1485.56   192.5  1491.5   202.1 1497.23
#Mann= 3 , 0 , 0
       0      .1       0    83.5    .045       0   105.9      .1       0
Bank Sta=83.5,105.9
XS Rating Curve= 0 ,0
Exp/Cntr=0.3,0.1

Type RM Length L Ch R = 1 ,5102.6  ,675.1,668,661
XS GIS Cut Line= 3
     1935114.136      356036.812     1935062.332      356101.568
     1935027.795      356317.421
#Sta/Elev= 25
       0 1469.73    18.4 1464.72    46.1 1457.05    55.3 1454.62    64.5  1452.7
    73.7 1451.23    82.9 1450.06    92.4 1449.12   111.4  1446.9     121 1445.69
     159 1440.55   167.8 1439.58     178 1438.97   187.5 1439.56     197  1441.6
   206.5 1443.86     216 1444.96   225.5  1445.7     235 1448.71   244.5 1456.45
     254 1467.86   263.5 1478.49     273 1486.03     292 1498.14   301.5 1504.12
#Mann= 3 , 0 , 0
       0      .1       0   167.8    .045       0   187.5      .1       0
Bank Sta=167.8,187.5
XS Rating Curve= 0 ,0
Exp/Cntr=0.3,0.1

Type RM Length L Ch R = 1 ,4434.6  ,604.6,612.7,620.8
XS GIS Cut Line= 3
     1934414.772      355993.642     1934393.187        356084.3
     1934427.724      356300.153
#Sta/Elev= 22
       0 1431.85     9.3 1428.95    74.6 1410.46    93.2 1405.03   102.7 1402.39
   112.2 1400.28   121.7 1399.65   131.2 1400.99   132.7 1401.48   140.7  1404.1
   150.2 1407.72   159.7 1410.89   169.2 1413.94   197.7 1423.66   216.8 1429.77
   235.8  1436.1   245.3 1439.45   254.8 1443.05   283.3 1454.38   292.8 1458.41
   302.3  1462.7   311.8 1467.12
#Mann= 3 , 0 , 0
       0      .1       0   112.2    .045       0   132.7      .1       0
Bank Sta=112.2,132.7
XS Rating Curve= 0 ,0
Exp/Cntr=0.3,0.1

Type RM Length L Ch R = 1 ,3821.9  ,535.1,513.9,492.5
XS GIS Cut Line= 2
     1933827.652      355985.007     1933784.481      356196.543
#Sta/Elev= 26
       0 1378.33     9.8 1378.02    19.6 1377.65    29.4 1377.25    39.2 1376.69
    49.1 1375.46    58.9 1373.24    68.7 1370.54    78.5 1367.81    88.3 1365.01
    97.7 1361.94    98.1 1361.81  102.461360.238     108 1358.24   112.7 1357.06
   117.8 1355.78   127.6 1356.33   137.4 1361.41   147.2 1369.19     157 1376.34
   166.8 1382.35   176.6 1387.78   186.5 1392.59   196.3 1396.29   206.1 1398.64
   215.9 1399.86
#Mann= 3 , 0 , 0
       0      .1       0  102.46    .045       0   127.6      .1       0
Bank Sta=102.46,127.6
XS Rating Curve= 0 ,0
Exp/Cntr=0.3,0.1
